HEC-RAS study H110-00-00.PRJ: H110-00-00

--- H110-00-00.g01 (geometry) --- (continued)

Type RM Length L Ch R = 3 ,2466.9,,,
BEGIN DESCRIPTION:
BUNTE STREET
Structure ID: H10-8
END DESCRIPTION:
Bridge Culvert--1,0,-1,-1, 0
Deck Dist Width WeirC Skew NumUp NumDn MinLoCord MaxHiCord MaxSubmerge Is_Ogee
10,31.6,2.6,, 46, 45,,,0.95,0,1,1,,
  4372.1  4392.1  4397.1  4407.1  4412.1  4447.1  4487.1  4527.1  4547.1  4562.1
    4600  4662.1  4671.3  4696.3  4706.3  4756.3  4770.9  4797.3  4837.2  4871.7
  4912.7  4982.1 4982.21  4982.3 5018.09  5018.2    5064  5101.4  5149.3  5192.9
  5195.3  5196.2  5251.2  5688.1  5703.1  5738.1  5753.1  5803.1  5818.1  6103.1
  6118.1  6123.1  6138.1  6153.1  6168.1  6368.1
   43.52   43.22   42.97   42.18   41.95   42.38   42.36   43.03   42.51   42.74
   42.33    42.4   42.42   42.46   42.47   42.55   42.58   42.62   42.49   42.38
   42.17   42.22   42.22   42.22   42.25   42.25    42.3   42.31   42.46   42.52
   42.52   42.52    42.5   42.34   42.81   42.32   42.72   43.43   42.71   42.93
   42.06   42.01   42.31   43.39   42.76   44.05
   43.52   43.22   42.97   42.18   41.95   42.38   42.36   43.03   42.51   42.74
   42.32   41.63   41.32   41.53   41.92   41.47   42.49   41.85   41.82   41.39
   41.12   40.01   40.01   41.22   41.25   39.61   41.17   41.67   41.48   41.75
   41.77   41.85   41.94   42.27    42.8   42.12   42.71   43.43   42.71   42.93
   42.06   42.01   42.31   43.39   42.76   44.05
  4372.1  4392.1  4397.1  4407.1  4412.1  4447.1  4487.1  4527.1  4547.1  4562.1
    4600  4662.1  4671.3  4696.3  4706.3  4756.3  4770.9  4797.3  4837.2  4871.7
  4911.4 4982.21  4982.3 5018.09  5018.2    5064  5101.4  5149.3  5192.9  5195.3
  5196.2  5251.2  5688.1  5703.1  5738.1  5753.1  5803.1  5818.1  6103.1  6118.1
  6123.1  6138.1  6153.1  6168.1  6368.1
   43.76   43.46   43.21   42.42   42.19   42.62    42.6   43.27   42.75   42.98
   42.56    42.4   42.42   42.46   42.47   42.55   42.73   42.62   42.49   42.38
   42.17   42.22   42.22   42.25   42.25    42.3   42.31   42.46   42.52   42.52
   42.52    42.5   42.51   43.04   42.36   42.95   43.67   42.95   43.17    42.3
   42.25   42.55   43.63      43   44.29
   43.76   43.46   43.21   42.42   42.19   42.62    42.6   43.27   42.75   42.98
   42.56   41.87   41.56   41.77   42.16   41.71   42.73   42.09   42.06   41.63
   41.37   40.25   41.46   41.49   39.85   41.41   41.91   41.72   41.99   42.01
   42.09   42.18   42.51   43.04   42.36   42.95   43.67   42.95   43.17    42.3
   42.25   42.55   43.63      43   44.29
Pier Skew, UpSta & Num, DnSta & Num=,4991.7, 2 ,4991.7, 2 , 0 , 0 , 0 ,,
       1       1
   35.15   42.23
       1       1
   35.39   42.47
Pier Skew, UpSta & Num, DnSta & Num=,5006.5, 2 ,5006.5, 2 , 0 , 0 , 0 ,,
       1       1
   34.43   42.24
       1       1
   34.66   42.48
Abutment Skew #Up #Dn=, 2 , 2
 4982.10 4994.70
   41.22   34.98
 4982.10 4994.70
   41.46   35.22
Abutment Skew #Up #Dn=, 2 , 2
 5005.50 5018.29
   35.10   41.25
 5005.50 5018.29
   35.34   41.49
BR Coef= 1 , 1 , 0 ,1.25, 0 ,,,0.8,0,2,0,
Wspro=,,,, 1 ,,,, 0 ,,,, 0 ,,,,-1 ,-1 ,-1 , 0 , 0 , 0 , 0 , 0
BC Design=,, 0 ,, 0 ,,,,,,
BR U #Sta/Elev= 79
  4372.1   43.52  4392.1   43.22  4397.1   42.97  4407.1   42.18  4412.1   41.95
  4447.1   42.38  4487.1   42.36  4527.1   43.03  4547.1   42.51  4562.1   42.74
    4600   42.32  4662.1   41.63    4667   41.46  4671.3   41.32  4696.3   41.53
  4706.3   41.92  4756.3   41.47  4770.9   42.49  4796.8   41.86  4797.3   41.85
  4835.2   41.82  4837.2   41.82  4871.7   41.39  4872.9   41.38  4911.4   41.13
  4912.7   41.12  4982.1   40.01 4982.21   40.01  4982.3   40.01 4983.29   39.99
  4983.4   39.99 4983.51   39.99  4984.1   39.98  4990.6   36.89  4991.7   36.38
  4994.6   35.03  4994.7   34.98  4994.9   35.06  4995.8   31.24  4999.2   30.91
    5004   31.25    5005   35.11  5005.4    35.1  5005.5    35.1  5006.5   35.75
  5010.6   37.29  5017.2   39.58 5018.09   39.61  5018.2   39.61  5018.3   39.62
 5019.49   39.66  5019.6   39.66 5019.71   39.67    5061   41.07    5064   41.17
  5101.4   41.67  5101.5   41.67  5148.5   41.48  5149.3   41.48  5192.9   41.75
  5195.3   41.77  5196.2   41.85  5251.2   41.94  5313.1   41.99  5325.1      42
  5688.1   42.27  5703.1    42.8  5738.1   42.12  5753.1   42.71  5800.8    43.4
  5803.1   43.43  5818.1   42.71  6103.1   42.93  6118.1   42.06  6123.1   42.01
  6138.1   42.31  6153.1   43.39  6168.1   42.76  6368.1   44.05
BR U #Mann= 5
 4372.10     0.2    4667     0.1  4984.1    0.02  5017.2     0.1  5325.1     0.2
BR U Banks=4984.10,5017.20
BR D #Sta/Elev= 79
  4372.1   43.76  4392.1   43.46  4397.1   43.21  4407.1   42.42  4412.1   42.19
  4447.1   42.62  4487.1    42.6  4527.1   43.27  4547.1   42.75  4562.1   42.98
    4600   42.56  4662.1   41.87    4667    41.7  4671.3   41.56  4696.3   41.77
  4706.3   42.16  4756.3   41.71  4770.9   42.73  4796.8    42.1  4797.3   42.09
  4835.2   42.06  4837.2   42.06  4871.7   41.63  4872.9   41.62  4911.4   41.37
  4912.7   41.36  4982.1   40.25 4982.21   40.25  4982.3   40.25 4983.29   40.23
  4983.4   40.23 4983.51   40.23  4984.1   40.22  4990.6   37.13  4991.7   36.62
  4994.6   35.27  4994.7   35.22  4994.9    35.3  4995.8   31.48  4999.2   31.15
    5004   31.49    5005   35.35  5005.4   35.34  5005.5   35.34  5006.5   35.99
  5010.6   37.53  5017.2   39.82 5018.09   39.85  5018.2   39.85  5018.3   39.86
 5019.49    39.9  5019.6    39.9 5019.71   39.91    5061   41.31    5064   41.41
  5101.4   41.91  5101.5   41.91  5148.5   41.72  5149.3   41.72  5192.9   41.99
  5195.3   42.01  5196.2   42.09  5251.2   42.18  5313.1   42.23  5325.1   42.24
  5688.1   42.51  5703.1   43.04  5738.1   42.36  5753.1   42.95  5800.8   43.64
  5803.1   43.67  5818.1   42.95  6103.1   43.17  6118.1    42.3  6123.1   42.25
  6138.1   42.55  6153.1   43.63  6168.1      43  6368.1   44.29
BR D #Mann= 5
 4372.10     0.2    4667     0.1  4984.1    0.02  5017.2     0.1  5325.1     0.2
BR D Banks=4984.10,5017.20

Type RM Length L Ch R = 1 ,2441.1,49.4,49.4,49.4
XS GIS Cut Line= 6
      3136366.29     13857511.19      3136644.40     13857657.85
      3136853.72     13857666.37      3136970.75     13857670.52
      3137262.45     13857681.18      3138229.58     13857239.75
BEGIN DESCRIPTION:
Downstream Section of Bridge/Culvert/Weir
END DESCRIPTION:
#Sta/Elev= 30
  4372.1   43.69  4392.1   43.39  4412.1   42.12  4527.1    43.2    4667   41.63
  4706.3   42.09  4756.3   41.64  4770.9   42.66  4797.3   42.02  4984.1   40.15
  4994.9   35.23  4995.8   31.41  4999.2   31.08    5004   31.42    5005   35.28
  5017.2   39.75    5064   41.34  5101.4   41.84  5325.1   42.17  5688.1   42.44
  5703.1   42.97  5738.1   42.29  5803.1    43.6  5818.1   42.88  6103.1    43.1
  6123.1   42.18  6138.1   42.48  6153.1   43.56  6168.1   42.93  6368.1   44.22
#Mann= 5 , 1 , 0
 4372.10     0.2       0    4667     0.1       0  4984.1    0.02       0
  5017.2     0.1       0  5325.1     0.2       0
#XS Ineff= 2 , 0
       0    4972      42    5025       0      42
Bank Sta=4984.10,5017.20
Exp/Cntr=0.5,0.3

Type RM Length L Ch R = 1 ,2391.7,508.9,515.6,516.8
XS GIS Cut Line= 3
      3136617.73     13857717.88      3137237.72     13857721.55
      3138217.22     13857273.99
BEGIN DESCRIPTION:
Cross Section 2391.7 - Interpolated
END DESCRIPTION:
#Sta/Elev= 25
    4667   43.25    4837   41.88    4967   41.16    4977   40.28 4984.09   39.87
 4988.29   37.99 4994.59   35.07 4995.19   31.12 5002.79   31.03 5005.19   31.38
 5005.39    35.1 5010.19   37.45 5016.49   39.92    5027    40.6    5037   41.02
    5287   41.93  5325.1    42.1  5413.9    42.5  5713.9   42.08  5723.9   42.75
  6143.9   42.49  6173.9   43.36  6193.9   42.46  6223.9   43.49  6363.9   43.41
#Mann= 5 , 1 , 0
 4667.00     0.2       0    4667     0.1       0 4984.09    0.02       0
 5016.49     0.1       0  5325.1     0.2       0
Bank Sta=4984.09,5016.49
Exp/Cntr=0.3,0.1

Type RM Length L Ch R = 1 ,1876.1,61.7,64.8,65
XS GIS Cut Line= 4
      3136526.02     13858110.42      3136790.15     13858202.13
      3137329.43     13858216.81      3138297.93     13857926.99
BEGIN DESCRIPTION:
Cross Section 1876.1 - Interpolated
END DESCRIPTION:
#Sta/Elev= 30
  4452.1   42.23  4561.7   42.55  4591.7   41.51  4641.7   42.14  4668.5   41.99
  4731.7   41.65  4811.2   42.01  4851.2   45.23  4881.2   46.52  4901.2   46.41
  4977.3   41.21  4985.8   37.05  4992.8   34.26  4995.3   30.57  5005.8    30.5
  5007.2   34.27  5014.6   39.51  5021.2   39.47  5041.2   41.52  5270.3   41.86
  5322.1   42.86  5562.1   41.86  5572.1   42.45  5592.1   41.48  5612.1   42.27
  5972.1   41.92  5992.1   42.52  6022.1   41.68  6032.1   42.28  6282.1   43.22
#Mann= 5 , 1 , 0
 4452.10     0.2       0  4668.5     0.1       0  4977.3    0.02       0
  5014.6     0.1       0  5270.3     0.2       0
Bank Sta=4977.30,5014.60
Exp/Cntr=0.5,0.3

Type RM Length L Ch R = 1 ,1811.3,43.4,43.4,43.4
XS GIS Cut Line= 6
      3135817.06     13857827.99      3136768.43     13858251.83
      3137083.50     13858267.42      3137328.72     13858279.15
      3138219.91     13857991.76      3138420.66     13857923.47
BEGIN DESCRIPTION:
Upstream Section of Bridge/Culvert/Weir
END DESCRIPTION:
#Sta/Elev= 30
  3640.7   43.43  3850.7   42.64  4015.7   43.71  4190.7   41.78  4215.7    42.7
  4260.7   41.84  4405.7   42.54  4605.7   42.39  4668.5   41.36  4743.3   40.61
  4743.5   41.75  4834.1   40.16    4900   39.98  4963.9    40.1  4977.3   41.14
  4992.8   34.19  4995.3    30.5  5005.8   30.43  5007.2    34.2  5014.6   39.44
  5072.2   40.77  5121.8   40.38  5238.5   41.08  5270.3   41.97  5951.6   42.15
  5971.6   42.83  6156.6   42.26  6301.6   43.63  6371.6   43.22  6391.6    43.9
#Mann= 5 , 1 , 0
 3640.70     0.2       0  4668.5     0.1       0  4977.3    0.02       0
  5014.6     0.1       0  5270.3     0.2       0
#XS Ineff= 2 , 0
       0    4972    41.7    5033       0      42
Bank Sta=4977.30,5014.60
Exp/Cntr=0.5,0.3

Type RM Length L Ch R = 3 ,1789.6,,,
BEGIN DESCRIPTION:
BRIDGE RAND STREET
Structure ID: H10-6
END DESCRIPTION:
Bridge Culvert--1,0,-1,-1, 0
Deck Dist Width WeirC Skew NumUp NumDn MinLoCord MaxHiCord MaxSubmerge Is_Ogee
10,23.4,2.6,, 55, 55,,,0.95,0,1,1,,
  3640.7  3715.7  3835.7  3850.7  3990.7  4015.7  4190.7  4215.7  4240.7  4260.7
  4305.7  4405.7  4425.7  4440.7  4465.7  4495.7  4520.7  4605.7  4635.7  4668.5
  4672.6  4688.3  4717.6  4723.3  4733.3  4738.3  4743.3  4743.5  4747.6    4769
  4834.1    4900  4963.9  4977.3 4982.21  4982.3 5022.19  5022.3  5022.4  5072.2
  5121.8  5184.4  5238.5  5260.1  5270.3  5271.6  5541.6  5951.6  5971.6  6001.6
  6081.6  6156.6  6301.6  6371.6  6391.6
   43.42   43.52   43.07   42.63   43.07    43.7   41.77   42.69   42.58   41.83
   41.85   42.53   42.08   42.33   41.96   42.36   41.85   42.38   42.22    41.6
    41.8   41.99    41.7   41.74   41.78   41.65   41.51   41.74   41.66   42.29
   42.18   42.32   42.51   42.46   42.44   42.44   42.41   42.41   42.41    42.3
      42   42.05   42.19   41.99   41.96   42.02   41.88   42.14   42.82   42.36
    42.6   42.25   43.62   43.21   43.89
   43.42   43.52   43.07   42.63   43.07    43.7   41.77   42.69   42.58   41.83
   41.85   42.53   42.08   42.33   41.96   42.36   41.85   42.38   42.22   41.35
   41.27   41.06   40.85   40.81   41.14   41.02    40.6   41.74   41.66   41.27
   40.15   39.97   40.09   41.13   38.73   40.58   40.55   39.61   39.61   40.76
   40.37   40.79   41.07    41.5   41.96   42.02   41.88   42.14   42.82   42.36
    42.6   42.25   43.62   43.21   43.89
  3640.7  3715.7  3835.7  3850.7  3990.7  4015.7  4190.7  4215.7  4240.7  4260.7
  4305.7  4405.7  4425.7  4440.7  4465.7  4495.7  4520.7  4605.7  4635.7  4668.5
  4672.6  4688.3  4717.6  4723.3  4733.3  4738.3  4743.3  4743.5  4747.6    4769
  4834.1    4900  4963.9  4977.3 4982.21  4982.3 5022.19  5022.3  5022.4  5072.2
  5121.8  5184.4  5238.5  5260.1  5270.3  5271.6  5541.6  5951.6  5971.6  6001.6
  6081.6  6156.6  6301.6  6371.6  6391.6
   43.38   43.48   43.03   42.59   43.03   43.66   41.73   42.65   42.54   41.79
   41.81   42.49   42.04   42.29   41.92   42.32   41.81   42.34   42.18    41.6
    41.8   41.99    41.7   41.74   41.78   41.65   41.51   41.71   41.63   42.29
   42.18   42.32   42.51   42.46   42.44   42.44   42.41   42.41   42.41    42.3
      42   42.05   42.19   41.99   41.93   41.98   41.84    42.1   42.78   42.32
   42.56   42.21   43.58   43.17   43.85
   43.34   43.44   42.99   42.55   42.99   43.62   41.69   42.61    42.5   41.75
   41.77   42.45      42   42.25   41.88   42.28   41.77    42.3   42.14   41.27
   41.19   40.98   40.77   40.73   41.06   40.94   40.52   41.66   41.58   41.19
   40.07   39.89   40.01   41.05   38.65    40.5   40.47   39.53   39.53   40.68
   40.29   40.71   40.99   41.42   41.88   41.94    41.8   42.06   42.74   42.28
   42.52   42.17   43.54   43.13   43.81
Pier Skew, UpSta & Num, DnSta & Num=,4990.7, 2 ,4990.7, 2 , 0 , 0 , 0 ,,
       1       1
   33.66   41.57
       1       1
   33.58   41.49
Pier Skew, UpSta & Num, DnSta & Num=,5010.0, 2 ,5010.0, 2 , 0 , 0 , 0 ,,
       1       1
   34.87   41.56
       1       1
   34.79   41.48
Abutment Skew #Up #Dn=, 2 , 2
 4982.10 4992.20
   40.58   34.24
 4982.10 4992.20
   40.50   34.16
Abutment Skew #Up #Dn=, 2 , 2
 5007.60 5022.39
   34.35   40.55
 5007.60 5022.39
   34.27   40.47
BR Coef= 1 , 1 , 0 ,1.25, 0 ,,,0.8,0,2,0,
Wspro=,,,, 1 ,,,, 0 ,,,, 0 ,,,,-1 ,-1 ,-1 , 0 , 0 , 0 , 0 , 0
BC Design=,, 0 ,, 0 ,,,,,,
BR U #Sta/Elev= 89
  3640.7   43.42  3715.7   43.52  3835.7   43.07  3850.7   42.63  3990.7   43.07
  4015.7    43.7  4190.7   41.77  4215.7   42.69  4240.7   42.58  4260.7   41.83
  4305.7   41.85  4405.7   42.53  4425.7   42.08  4440.7   42.33  4465.7   41.96
  4495.7   42.36  4520.7   41.85  4605.7   42.38  4635.7   42.22  4668.5   41.35
  4670.7   41.29  4672.6   41.27  4687.6   41.07  4688.3   41.06  4717.6   40.85
  4723.3   40.81  4732.6   41.12  4733.3   41.14  4738.3   41.02  4743.3    40.6
  4743.5   41.74  4747.6   41.66    4769   41.27  4770.4   41.24  4833.6   40.16
  4834.1   40.15    4900   39.97  4901.3   39.97  4963.9   40.09  4965.2   40.19
 4976.39   41.06  4976.5   41.07 4976.61   41.08  4977.3   41.13  4982.1   38.78
 4982.21   38.73  4982.3   38.68  4985.8   36.97  4990.7   34.87  4992.1   34.28
  4992.2   34.24  4992.8   34.18  4995.3   30.49  5000.5   30.45  5005.8   30.42
  5007.2   34.19  5007.5   34.27  5007.6   34.35    5010   36.27  5011.7   37.27
  5014.6   39.43 5022.19   39.61  5022.3   39.61  5022.4   39.61 5028.99   39.76
  5029.1   39.76 5029.21   39.77  5072.2   40.76    5073   40.75  5121.8   40.37
  5122.8   40.38  5183.7   40.79  5184.4   40.79  5238.4   41.07  5238.5   41.07
  5260.1    41.5  5270.3   41.96  5271.6   42.02  5401.6   41.97  5541.6   41.88
  5571.6   41.91  5951.6   42.14  5971.6   42.82  6001.6   42.36  6081.6    42.6
  6156.6   42.25  6301.6   43.62  6371.6   43.21  6391.6   43.89
BR U #Mann= 5
 3640.70     0.2  4668.5     0.1  4977.3    0.02  5014.6     0.1  5270.3     0.2
BR U Banks=4977.30,5014.60
BR D #Sta/Elev= 89
  3640.7   43.34  3715.7   43.44  3835.7   42.99  3850.7   42.55  3990.7   42.99
  4015.7   43.62  4190.7   41.69  4215.7   42.61  4240.7    42.5  4260.7   41.75
  4305.7   41.77  4405.7   42.45  4425.7      42  4440.7   42.25  4465.7   41.88
  4495.7   42.28  4520.7   41.77  4605.7    42.3  4635.7   42.14  4668.5   41.27
  4670.7   41.21  4672.6   41.19  4687.6   40.99  4688.3   40.98  4717.6   40.77
  4723.3   40.73  4732.6   41.04  4733.3   41.06  4738.3   40.94  4743.3   40.52
  4743.5   41.66  4747.6   41.58    4769   41.19  4770.4   41.16  4833.6   40.08
  4834.1   40.07    4900   39.89  4901.3   39.89  4963.9   40.01  4965.2   40.11
 4976.39   40.98  4976.5   40.99 4976.61      41  4977.3   41.05  4982.1    38.7
 4982.21   38.65  4982.3    38.6  4985.8   36.89  4990.7   34.79  4992.1    34.2
  4992.2   34.16  4992.8    34.1  4995.3   30.41  5000.5   30.37  5005.8   30.34
  5007.2   34.11  5007.5   34.19  5007.6   34.27    5010   36.19  5011.7   37.19
  5014.6   39.35 5022.19   39.53  5022.3   39.53  5022.4   39.53 5028.99   39.68
  5029.1   39.68 5029.21   39.69  5072.2   40.68    5073   40.67  5121.8   40.29
  5122.8    40.3  5183.7   40.71  5184.4   40.71  5238.4   40.99  5238.5   40.99
  5260.1   41.42  5270.3   41.88  5271.6   41.94  5401.6   41.89  5541.6    41.8
  5571.6   41.83  5951.6   42.06  5971.6   42.74  6001.6   42.28  6081.6   42.52
  6156.6   42.17  6301.6   43.54  6371.6   43.13  6391.6   43.81
BR D #Mann= 5
 3640.70     0.2  4668.5     0.1  4977.3    0.02  5014.6     0.1  5270.3     0.2
BR D Banks=4977.30,5014.60

Type RM Length L Ch R = 1 ,1767.9,11.8,11.8,11.8
XS GIS Cut Line= 6
      3135834.78     13857867.61      3136786.15     13858291.45
      3137101.22     13858307.04      3137346.44     13858318.77
      3138237.63     13858031.38      3138438.38     13857963.09
BEGIN DESCRIPTION:
Downstream Section of Bridge/Culvert/Weir
END DESCRIPTION:
#Sta/Elev= 30
  3640.7   43.38  3850.7   42.59  4015.7   43.66  4190.7   41.73  4215.7   42.65
  4260.7   41.79  4405.7   42.49  4605.7   42.34  4668.5   41.31  4743.3   40.56
  4743.5    41.7  4834.1   40.11    4900   39.93  4963.9   40.05  4977.3   41.09
  4992.8   34.14  4995.3   30.45  5005.8   30.38  5007.2   34.15  5014.6   39.39
  5072.2   40.72  5121.8   40.33  5238.5   41.03  5270.3   41.92  5951.6    42.1
  5971.6   42.78  6156.6   42.21  6301.6   43.58  6371.6   43.17  6391.6   43.85
#Mann= 5 , 1 , 0
 3640.70     0.2       0  4668.5     0.1       0  4977.3    0.02       0
  5014.6     0.1       0  5270.3     0.2       0
#XS Ineff= 2 , 0
       0    4972    41.5    5033       0    41.8
Bank Sta=4977.30,5014.60
Exp/Cntr=0.5,0.3

Type RM Length L Ch R = 3 ,1766.6,,,
BEGIN DESCRIPTION:
Pipeline
END DESCRIPTION:
Bridge Culvert--1,0,-1,-1, 0
Deck Dist Width WeirC Skew NumUp NumDn MinLoCord MaxHiCord MaxSubmerge Is_Ogee
10,1,2.6,, 60, 60,,,0.95,0,1,1,,
  4461.3  4491.3  4521.3  4551.3  4626.3  4686.3  4716.3  4836.3  4851.2  4866.2
  4876.2  4911.2 4920.45 4925.35 4928.05 4963.15 4975.15 4980.95 5024.15 5025.84
 5025.95 5026.05 5063.25 5066.95  5136.2  5196.2  5217.6  5242.6  5272.6    5320
    5405    5420    5435    5455    5470    5605    5615    5650    5700    5745
    5825    5865    5890    5895    5905    5910    5925    5955    5980    6000
    6015  6030.6  6120.6  6285.6  6300.6  6330.6  6335.6  6350.6  6380.6  6421.6
   44.38    43.2   43.03   41.75   41.21   41.29    41.9   40.72   41.01   40.89
   40.27   40.52   42.11   42.14   39.99   40.34   39.65      42   42.23   41.01
   40.93   39.65   41.67    41.5   41.07   41.32   41.79   41.89   41.54   41.91
   42.04   41.74   41.96   41.84   42.48   42.23   42.38    41.9   41.84   41.28
   42.14   42.27   41.68   41.83   42.76   42.97   42.13   42.91   42.97   44.28
   44.31   43.41   42.38   42.98   42.41   43.85   43.75   42.78   43.34   43.16
   44.38    43.2   43.03   41.75   41.21   41.29    41.9   40.72   41.01   40.89
   40.27   40.52   42.11   42.14   39.99   40.34   39.64   41.33   41.56   40.34
   39.65   39.65   41.67    41.5   41.07   41.32   41.79   41.89   41.54   41.91
   42.04   41.74   41.96   41.84   42.48   42.23   42.38    41.9   41.84   41.28
   42.14   42.27   41.68   41.83   42.76   42.97   42.13   42.91   42.97   44.28
   44.31   43.41   42.38   42.98   42.41   43.85   43.75   42.78   43.34   43.16
  4461.3  4491.3  4521.3  4551.3  4626.3  4686.3  4716.3  4836.3  4851.2  4866.2
  4876.2  4911.2 4920.45 4925.35 4928.05 4963.15 4975.15 4980.95 5024.15 5025.84
 5025.95 5026.05 5063.25 5066.95  5136.2  5196.2  5217.6  5242.6  5272.6    5320
    5405    5420    5435    5455    5470    5605    5615    5650    5700    5745
    5825    5865    5890    5895    5905    5910    5925    5955    5980    6000
    6015  6030.6  6120.6  6285.6  6300.6  6330.6  6335.6  6350.6  6380.6  6421.6
   44.38    43.2   43.03   41.75   41.21   41.29    41.9   40.72   41.01   40.89
   40.27   40.52   42.11   42.14   39.99   40.34   39.65      42   42.23   41.01
   40.93   39.65   41.67    41.5   41.07   41.32   41.79   41.89   41.54   41.91
   42.04   41.74   41.96   41.84   42.48   42.23   42.38    41.9   41.84   41.28
   42.14   42.27   41.68   41.83   42.76   42.97   42.13   42.91   42.97   44.28
   44.31   43.41   42.38   42.98   42.41   43.85   43.75   42.78   43.34   43.16
   44.38    43.2   43.03   41.75   41.21   41.29    41.9   40.72   41.01   40.89
   40.27   40.52   42.11   42.14   39.99   40.34   39.64   41.33   41.56   40.34
   39.65   39.65   41.67    41.5   41.07   41.32   41.79   41.89   41.54   41.91
   42.04   41.74   41.96   41.84   42.48   42.23   42.38    41.9   41.84   41.28
   42.14   42.27   41.68   41.83   42.76   42.97   42.13   42.91   42.97   44.28
   44.31   43.41   42.38   42.98   42.41   43.85   43.75   42.78   43.34   43.16
BR Coef= 1 , 1 , 0 ,1.25, 0 ,,,0.8,0,2,0,
Wspro=,,,, 1 ,,,, 0 ,,,, 0 ,,,,-1 ,-1 ,-1 , 0 , 0 , 0 , 0 , 0
BC Design=,, 0 ,, 0 ,,,,,,
BR U #Sta/Elev= 75
  4461.3   44.38  4491.3    43.2  4521.3   43.03  4551.3   41.75  4626.3   41.21
  4686.3   41.29  4716.3    41.9  4766.3   41.34  4836.3   40.72  4851.2   41.01
  4866.2   40.89  4876.2   40.27  4911.2   40.52 4920.45   42.11 4925.35   42.14
 4928.05   39.99 4963.15   40.34 4974.95   39.65 4975.06   39.65 4975.15   39.64
 4980.95    39.3 4983.95   39.13 4989.95   36.55 4993.75   34.59 4994.55   30.38
 4995.85   30.42 5005.95   30.85 5012.35   37.37 5016.05   39.14 5021.85   39.44
 5024.15   39.56 5025.84   39.64 5025.95   39.65 5026.05   39.65 5060.05   41.38
 5063.25   41.67 5066.95    41.5  5136.2   41.07  5196.2   41.32  5217.6   41.79
  5242.6   41.89  5272.6   41.54    5320   41.91    5405   42.04    5420   41.74
    5435   41.96    5455   41.84    5470   42.48    5605   42.23    5615   42.38
    5650    41.9    5700   41.84    5745   41.28    5825   42.14    5865   42.27
    5890   41.68    5895   41.83    5905   42.76    5910   42.97    5925   42.13
    5955   42.91    5980   42.97    6000   44.28    6015   44.31  6015.6   44.27
  6030.6   43.41  6120.6   42.38  6285.6   42.98  6300.6   42.41  6330.6   43.85
  6335.6   43.75  6345.6   42.97  6350.6   42.78  6380.6   43.34  6421.6   43.16
BR U #Mann= 4
 4461.30     0.1 4983.95    0.02 5016.05     0.1  6421.6     0.2
BR U Banks=4983.95,5016.05
BR D #Sta/Elev= 75
  4461.3   44.38  4491.3    43.2  4521.3   43.03  4551.3   41.75  4626.3   41.21
  4686.3   41.29  4716.3    41.9  4766.3   41.34  4836.3   40.72  4851.2   41.01
  4866.2   40.89  4876.2   40.27  4911.2   40.52 4920.45   42.11 4925.35   42.14
 4928.05   39.99 4963.15   40.34 4974.95   39.65 4975.06   39.65 4975.15   39.64
 4980.95    39.3 4983.95   39.13 4989.95   36.55 4993.75   34.59 4994.55   30.38
 4995.85   30.42 5005.95   30.85 5012.35   37.37 5016.05   39.14 5021.85   39.44
 5024.15   39.56 5025.84   39.64 5025.95   39.65 5026.05   39.65 5060.05   41.38
 5063.25   41.67 5066.95    41.5  5136.2   41.07  5196.2   41.32  5217.6   41.79
  5242.6   41.89  5272.6   41.54    5320   41.91    5405   42.04    5420   41.74
    5435   41.96    5455   41.84    5470   42.48    5605   42.23    5615   42.38
    5650    41.9    5700   41.84    5745   41.28    5825   42.14    5865   42.27
    5890   41.68    5895   41.83    5905   42.76    5910   42.97    5925   42.13
    5955   42.91    5980   42.97    6000   44.28    6015   44.31  6015.6   44.27
  6030.6   43.41  6120.6   42.38  6285.6   42.98  6300.6   42.41  6330.6   43.85
  6335.6   43.75  6345.6   42.97  6350.6   42.78  6380.6   43.34  6421.6   43.16
BR D #Mann= 4
 4461.30     0.1 4983.95    0.02 5016.05     0.1  6421.6     0.2
BR D Banks=4983.95,5016.05

Type RM Length L Ch R = 1 ,1756.1,219.4,219.4,219.4
XS GIS Cut Line= 6
      3136576.23     13858327.63      3136966.06     13858327.63
      3137332.29     13858339.44      3137434.68     13858339.44
      3138127.76     13858280.37      3138509.74     13858142.54
BEGIN DESCRIPTION:
Downstream Section of Bridge/Culvert/Weir
END DESCRIPTION:
#Sta/Elev= 30
  4461.3   44.38  4551.3   41.75  4626.3   41.21  4716.3    41.9  4876.2   40.27
  4911.2   40.52 4925.35   42.14 4928.05   39.99 4963.15   40.34 4983.95   39.13
 4993.75   34.59 4994.55   30.38 5005.95   30.85 5012.35   37.37 5016.05   39.14
 5063.25   41.67  5136.2   41.07    5470   42.48    5745   41.28    5865   42.27
    5890   41.68    5910   42.97    5925   42.13    6015   44.31  6030.6   43.41
  6120.6   42.38  6300.6   42.41  6330.6   43.85  6350.6   42.78  6421.6   43.16
#Mann= 4 , 1 , 0
 4461.30     0.1       0 4983.95    0.02       0 5016.05     0.1       0
  6421.6     0.2       0
#XS Ineff= 2 , 0
       0    4972    41.3    5033       0    41.6
Bank Sta=4983.95,5016.05
Exp/Cntr=0.5,0.3

Type RM Length L Ch R = 1 ,1536.7,379.9,399.9,412.2
XS GIS Cut Line= 2
      3136819.50     13858576.33      3137567.89     13858462.60
BEGIN DESCRIPTION:
Cross Section 1536.7 - Interpolated
END DESCRIPTION:
#Sta/Elev= 17
  4617.2   41.89  4954.2   41.35  4964.2   40.65  4974.2    39.4 4983.95   39.09
 4989.95   36.51 4993.75   34.55 4994.55   30.34 4995.85   30.38 5005.95   30.81
 5012.35   37.33 5016.05    39.1  5034.2   41.04  5054.2   42.39  5104.2   40.64
  5334.2   42.28  5374.2   42.02
#Mann= 3 , 1 , 0
 4617.20     0.1       0 4983.95    0.02       0 5016.05     0.1       0
Bank Sta=4983.95,5016.05
Exp/Cntr=0.3,0.1

Type RM Length L Ch R = 1 ,1136.8,115,114.8,105.9
XS GIS Cut Line= 2
      3136939.20     13858834.53      3137694.97     13858955.60
BEGIN DESCRIPTION:
Cross Section 1136.8 - Interpolated
END DESCRIPTION:
#Sta/Elev= 23
  4613.8    42.7  4619.2   42.26  4629.2   41.92  4701.5    41.7  4959.2   40.91
  4969.2   40.32  4983.5   39.38  4989.7   36.43  4994.1   34.28  4994.2   30.54
  4995.8   30.27  5005.5   30.46  5005.9   34.32  5012.6   35.61  5017.2   39.15
  5029.2   40.35  5039.2   41.65  5049.2   42.32  5089.2   40.92  5258.6   41.89
  5309.2   42.18  5319.2   41.89  5379.2   41.91
#Mann= 5 , 1 , 0
 4613.80     0.2       0  4701.5     0.1       0  4983.5    0.02       0
  5017.2     0.1       0  5258.6     0.2       0
Bank Sta=4983.50,5017.20
Exp/Cntr=0.5,0.3

Type RM Length L Ch R = 1 ,1022.0,24,24,24
XS GIS Cut Line= 6
      3136493.40     13858440.23      3137039.56     13858997.42
      3137285.81     13859009.15      3137651.74     13859023.81
      3138254.76     13858497.49      3138437.34     13858328.44
BEGIN DESCRIPTION:
Upstream Section of Bridge/Culvert/Weir
END DESCRIPTION:
#Sta/Elev= 30
  3935.2   46.13  4110.2   43.25  4145.2   41.04  4235.2   42.71  4435.2   41.77
  4460.2   43.35  4510.2   43.82  4545.2   42.14  4701.5   41.47  4814.2   42.06
  4967.7   40.41  4983.5   39.36  4989.7   36.41  4992.7   37.02  4994.1   34.26
  4994.2   30.52  4995.8   30.25  5005.5   30.44  5005.9    34.3  5012.6   35.59
  5017.2   39.13  5076.2   41.09  5258.6   42.23  5706.3   41.64  5796.3    42.9
  5816.3   42.02  6046.3   41.99  6316.3   42.49  6341.3   43.87  6377.4   43.16
#Mann= 5 , 1 , 0
 3935.20     0.2       0  4701.5     0.1       0  4983.5    0.02       0
  5017.2     0.1       0  5258.6     0.2       0
#XS Ineff= 2 , 0
       0    4975    39.8    5025       0    39.8
Bank Sta=4983.50,5017.20
Exp/Cntr=0.5,0.3

Type RM Length L Ch R = 3 ,1010.0,,,
BEGIN DESCRIPTION:
PARDEE STREET
Structure ID: H10-4
END DESCRIPTION:
Bridge Culvert--1,0,-1,-1, 0
Deck Dist Width WeirC Skew NumUp NumDn MinLoCord MaxHiCord MaxSubmerge Is_Ogee
10,4,2.6,, 60, 60,,,0.95,0,1,1,,
  3935.2  4000.2  4010.2  4025.2  4040.2  4110.2  4130.2  4145.2  4170.2  4235.2
  4305.2  4335.2  4350.2  4435.2  4460.2  4485.2  4510.2  4520.2  4530.2  4540.2
  4545.2  4700.2  4701.4  4708.1  4818.3  4864.3  4910.3  4915.7  4967.7  4983.5
    4986  4986.4  4986.5 5020.59  5020.8  5076.2  5134.4  5201.8  5247.2  5265.2
  5298.6  5313.6  5328.6  5356.3  5391.3  5431.3  5636.3  5681.3  5691.3  5706.3
  5776.3  5786.3  5796.3  5816.3  6021.3  6046.3  6316.3  6341.3  6361.3  6377.4
   46.13   45.56   45.25   44.31   44.49   43.25   41.65   41.04   41.75   42.71
   42.64   41.85   42.14   41.77   43.35   43.79   43.82   43.42   42.51   42.49
   42.14   41.51   41.96   41.97   42.12   41.77   41.27   41.21   40.42   39.98
   39.93   39.93   39.93   40.16   40.16   41.34   41.82   42.21   42.44   42.56
   41.79   42.08   41.54   42.11   41.83   42.28   41.66   42.46   42.34   41.64
    41.9   42.62    42.9   42.02   42.53   41.99   42.49   43.87   43.81   43.16
   46.13   45.56   45.25   44.31   44.49   43.25   41.65   41.04   41.75   42.71
   42.64   41.85   42.14   41.77   43.35   43.79   43.82   43.42   42.51   42.49
   42.14   41.51   41.47   41.26   41.95    40.7    40.3   40.64   40.41   39.36
   38.17   37.98   38.93   39.16   38.85   41.09   41.55   41.41   41.67   42.56
   41.79   42.08   41.54   42.11   41.83   42.28   41.66   42.46   42.34   41.64
    41.9   42.62    42.9   42.02   42.53   41.99   42.49   43.87   43.81   43.16
  3935.2  4000.2  4010.2  4025.2  4040.2  4110.2  4130.2  4145.2  4170.2  4235.2
  4305.2  4335.2  4350.2  4435.2  4460.2  4485.2  4510.2  4520.2  4530.2  4540.2
  4545.2  4700.2  4701.4  4708.1  4818.3  4864.3  4910.3  4915.7  4967.7  4983.5
    4986  4986.4  4986.5 5020.59  5020.8  5076.2  5134.4  5201.8  5247.2  5265.2
  5298.6  5313.6  5328.6  5356.3  5391.3  5431.3  5636.3  5681.3  5691.3  5706.3
  5776.3  5786.3  5796.3  5816.3  6021.3  6046.3  6316.3  6341.3  6361.3  6377.4
   46.13   45.56   45.25   44.31   44.49   43.25   41.65   41.04   41.75   42.71
   42.64   41.85   42.14   41.77   43.35   43.79   43.82   43.42   42.51   42.49
   42.14   41.51   41.96   41.97   42.12   41.77   41.27   41.21   40.42   39.98
   39.93   39.93   39.93   40.16   40.16   41.34   41.82   42.21   42.44   42.56
   41.79   42.08   41.54   42.11   41.83   42.28   41.66   42.46   42.34   41.64
    41.9   42.62    42.9   42.02   42.53   41.99   42.49   43.87   43.81   43.16
   45.96   45.39   45.08   44.14   44.32   43.08   41.48   40.87   41.58   42.54
   42.47   41.68   41.97    41.6   43.18   43.62   43.65   43.25   42.34   42.32
   41.97   41.34    41.3   41.09   41.78   40.53   40.13   40.47   40.24   39.19
      38   37.81   38.76   38.99   38.68   40.92   41.38   41.24    41.5   42.39
   41.62   41.91   41.37   41.94   41.66   42.11   41.49   42.29   42.17   41.47
   41.73   42.45   42.73   41.85   42.36   41.82   42.32    43.7   43.64   42.99
Pier Skew, UpSta & Num, DnSta & Num=,4992.7, 2 ,4992.7, 2 , 0 , 0 , 0 ,,
     0.5     0.5
   35.53   39.97
     0.5     0.5
   35.36    39.8
Pier Skew, UpSta & Num, DnSta & Num=,5012.6, 2 ,5012.6, 2 , 0 , 0 , 0 ,,
     0.5     0.5
   34.54   40.11
     0.5     0.5
   34.37   39.94
BR Coef= 1 , 1 , 0 ,1.25, 0 ,,,0.8,-1,2,0,
Wspro=,,,, 1 ,,,, 0 ,,,, 0 ,,,,-1 ,-1 ,-1 , 0 , 0 , 0 , 0 , 0
BC Design=,, 0 ,, 0 ,,,,,,
BR U #Sta/Elev= 99
  3935.2   46.13  4000.2   45.56  4010.2   45.25  4025.2   44.31  4040.2   44.49
  4075.2   43.71  4090.2   43.73  4110.2   43.25  4130.2   41.65  4145.2   41.04
  4170.2   41.75  4235.2   42.71  4245.2   42.69  4305.2   42.64  4335.2   41.85
  4350.2   42.14  4435.2   41.77  4440.2   41.91  4460.2   43.35  4480.2   43.56
  4485.2   43.79  4510.2   43.82  4520.2   43.42  4530.2   42.51  4540.2   42.49
  4545.2   42.14  4700.2   41.51  4701.4   41.47  4701.5   41.47  4708.1   41.26
  4814.2   42.06  4818.3   41.95  4864.3    40.7  4865.8   40.69  4910.3    40.3
  4915.7   40.64  4916.1   40.64  4967.7   40.41  4983.5   39.36    4986   38.17
 4986.11   38.12 4986.19   38.08  4986.3   38.03  4986.4   37.98  4986.5   37.93
 4986.61   37.88  4989.7   36.41  4992.7   37.02  4994.1   34.26  4994.2   30.52
  4995.8   30.25  5005.5   30.44  5005.9    34.3  5012.6   35.59  5017.2   39.13
  5020.2   38.83  5020.5   38.84 5020.59   38.85  5020.7   38.85  5020.8   38.85
 5021.09   38.87  5021.2   38.87 5021.31   38.87  5073.2   40.97  5076.2   41.09
  5134.4   41.55  5139.8   41.54  5201.6   41.41  5201.8   41.41  5247.2   41.67
  5248.9   41.75  5258.6   42.23  5265.2   42.56  5268.6   42.36  5298.6   41.79
  5313.6   42.08  5328.6   41.54  5331.3   41.54  5356.3   42.11  5391.3   41.83
  5431.3   42.28  5636.3   41.66  5681.3   42.46  5691.3   42.34  5706.3   41.64
  5741.3   41.92  5776.3    41.9  5786.3   42.62  5796.3    42.9  5816.3   42.02
  5931.3   42.16  5956.3    42.5  5966.3   42.25  6021.3   42.53  6046.3   41.99
  6316.3   42.49  6341.3   43.87  6361.3   43.81  6377.4   43.16
BR U #Mann= 5
 3935.20     0.2  4701.5     0.1  4983.5    0.02  5017.2     0.1  5258.6     0.2
BR U Banks=4983.50,5017.20
BR D #Sta/Elev= 99
  3935.2   45.96  4000.2   45.39  4010.2   45.08  4025.2   44.14  4040.2   44.32
  4075.2   43.54  4090.2   43.56  4110.2   43.08  4130.2   41.48  4145.2   40.87
  4170.2   41.58  4235.2   42.54  4245.2   42.52  4305.2   42.47  4335.2   41.68
  4350.2   41.97  4435.2    41.6  4440.2   41.74  4460.2   43.18  4480.2   43.39
  4485.2   43.62  4510.2   43.65  4520.2   43.25  4530.2   42.34  4540.2   42.32
  4545.2   41.97  4700.2   41.34  4701.4    41.3  4701.5    41.3  4708.1   41.09
  4814.2   41.89  4818.3   41.78  4864.3   40.53  4865.8   40.52  4910.3   40.13
  4915.7   40.47  4916.1   40.47  4967.7   40.24  4983.5   39.19    4986      38
 4986.11   37.95 4986.19   37.91  4986.3   37.86  4986.4   37.81  4986.5   37.76
 4986.61   37.71  4989.7   36.24  4992.7   36.85  4994.1   34.09  4994.2   30.35
  4995.8   30.08  5005.5   30.27  5005.9   34.13  5012.6   35.42  5017.2   38.96
  5020.2   38.66  5020.5   38.67 5020.59   38.68  5020.7   38.68  5020.8   38.68
 5021.09    38.7  5021.2    38.7 5021.31    38.7  5073.2    40.8  5076.2   40.92
  5134.4   41.38  5139.8   41.37  5201.6   41.24  5201.8   41.24  5247.2    41.5
  5248.9   41.58  5258.6   42.06  5265.2   42.39  5268.6   42.19  5298.6   41.62
  5313.6   41.91  5328.6   41.37  5331.3   41.37  5356.3   41.94  5391.3   41.66
  5431.3   42.11  5636.3   41.49  5681.3   42.29  5691.3   42.17  5706.3   41.47
  5741.3   41.75  5776.3   41.73  5786.3   42.45  5796.3   42.73  5816.3   41.85
  5931.3   41.99  5956.3   42.33  5966.3   42.08  6021.3   42.36  6046.3   41.82
  6316.3   42.32  6341.3    43.7  6361.3   43.64  6377.4   42.99
BR D #Mann= 5
 3935.20     0.2  4701.5     0.1  4983.5    0.02  5017.2     0.1  5258.6     0.2
BR D Banks=4983.50,5017.20

Type RM Length L Ch R = 1 ,998.0,1,1,1
XS GIS Cut Line= 6
      3136491.04     13858464.11      3137037.20     13859021.30
      3137283.45     13859033.03      3137649.38     13859047.69
      3138252.40     13858521.37      3138434.97     13858352.33
BEGIN DESCRIPTION:
Downstream Section of Bridge/Culvert/Weir
END DESCRIPTION:
#Sta/Elev= 30
  3935.2   46.06  4110.2   43.18  4145.2   40.97  4235.2   42.64  4435.2    41.7
  4460.2   43.28  4510.2   43.75  4545.2   42.07  4701.5    41.4  4814.2   41.99
  4967.7   40.34  4983.5   39.29  4989.7   36.34  4992.7   36.95  4994.1   34.19
  4994.2   30.45  4995.8   30.18  5005.5   30.37  5005.9   34.23  5012.6   35.52
  5017.2   39.06  5076.2   41.02  5258.6   42.16  5706.3   41.57  5796.3   42.83
  5816.3   41.95  6046.3   41.92  6316.3   42.42  6341.3    43.8  6377.4   43.09
#Mann= 5 , 1 , 0
 3935.20     0.2       0  4701.5     0.1       0  4983.5    0.02       0
  5017.2     0.1       0  5258.6     0.2       0
#XS Ineff= 2 , 0
       0    4975    39.7    5025       0    39.7
Bank Sta=4983.50,5017.20
Exp/Cntr=0.5,0.3

Type RM Length L Ch R = 1 ,997.0,417.6,424.7,429.3
XS GIS Cut Line= 2
      3136864.70     13859045.16      3137750.57     13859065.30
BEGIN DESCRIPTION:
Cross Section 997.0
END DESCRIPTION:
#Sta/Elev= 30
  4545.2   42.14  4701.5   41.47  4823.1   40.97  4833.1   40.47  4917.1   40.41
 4922.04   40.63 4967.04   40.14 4979.84    38.9 4982.54   39.17 4994.14   34.38
 4995.14   30.34 5004.04   30.18 5005.84   34.31 5007.44   34.19 5018.14   38.91
 5027.54   39.11 5037.34   40.03 5059.74   40.22 5089.24   39.73  5102.8   41.67
  5147.8   40.79  5233.6   41.44  5258.6   41.89  5268.6   42.36  5298.6   41.79
  5313.6   42.08  5331.3   41.54  5356.3   42.11  5391.3   41.83  5431.3   42.28
#Mann= 5 , 1 , 0
 4545.20     0.2       0  4701.5     0.1       0 4982.54    0.02       0
 5018.14     0.1       0  5258.6     0.2       0
Bank Sta=4982.54,5018.14
Exp/Cntr=0.3,0.1

Type RM Length L Ch R = 1 ,572.3,108.1,116,101.7
XS GIS Cut Line= 2
      3137135.00     13859420.10      3137534.87     13859478.79
BEGIN DESCRIPTION:
Cross Section 572.3 - Interpolated
END DESCRIPTION:
#Sta/Elev= 19
  4772.8   42.05  4846.9   42.01  4956.9   40.14  4966.9   39.17  4976.9   37.36
  4986.8   38.56  4991.4   35.98  4995.7    33.8  4995.9   30.05  5002.6   30.07
  5003.6   29.97  5004.3   33.74  5015.5   38.69  5016.9   37.61  5036.9   40.28
  5056.9   40.89  5146.9    41.8  5162.5    41.7  5176.9    41.6
#Mann= 4 , 1 , 0
 4772.80     0.1       0  4986.8    0.02       0  5015.5     0.1       0
  5162.5     0.2       0
Bank Sta=4986.80,5015.50
Exp/Cntr=0.5,0.3

Type RM Length L Ch R = 1 ,456.3,44.6,44.6,44.6
XS GIS Cut Line= 4
      3137022.28     13859474.34      3137187.91     13859557.61
      3137530.98     13859571.81      3137596.74     13859566.90
BEGIN DESCRIPTION:
Upstream Section of Bridge/Culvert/Weir
END DESCRIPTION:
#Sta/Elev= 27
  4597.9   41.63  4758.3    41.5  4802.8   41.47  4819.8   40.79  4853.8    41.1
  4890.9   41.24  4939.1   40.53  4966.2   40.03  4973.2   40.36  4983.9   41.27
  4986.8    38.5  4991.4   35.92  4995.7   33.74  4995.9   29.99  5002.6   30.01
  5003.6   29.91  5004.3   33.68  5015.5   38.63  5026.7   41.14  5028.7   41.29
  5044.7   41.26  5089.5   39.17  5095.2   40.99  5095.3   41.21  5119.4   41.53
  5162.5   41.67  5192.6   41.76
#Mann= 5 , 1 , 0
 4597.90     0.2       0  4758.3     0.1       0  4986.8    0.02       0
  5015.5     0.1       0  5162.5     0.2       0
#XS Ineff= 2 , 0
       0    4975    41.5    5030       0    41.5
Bank Sta=4986.80,5015.50
Exp/Cntr=0.5,0.3

Type RM Length L Ch R = 3 ,434.0,,,
BEGIN DESCRIPTION:
MIDEN STREET
Structure ID: H10-2
END DESCRIPTION:
Bridge Culvert--1,0,-1,-1, 0
Deck Dist Width WeirC Skew NumUp NumDn MinLoCord MaxHiCord MaxSubmerge Is_Ogee
10,24.6,2.6,,51,51,,,0.95,0,1,1,,
  4597.9  4758.3  4802.8  4819.6  4819.8  4851.8  4853.8  4888.2  4890.9  4939.1
  4941.2  4966.2  4973.2  4983.9 4984.51  4984.6  4984.7 4985.79  4985.9 4986.01
  4986.8  4990.6  4991.4  4995.7  4995.9  5002.6  5003.6  5004.3  5015.5  5019.6
 5019.69  5019.8  5026.7 5027.99  5028.1 5028.21  5028.6  5028.7  5044.4  5044.7
  5089.5  5095.2  5095.3  5095.4  5119.4  5144.2  5144.6  5162.5  5190.1  5190.4
  5192.6
   41.63    41.5   41.47   41.94   41.94   41.83   41.83   41.81    41.8   41.59
   41.58   41.53   41.52   41.49   41.49   41.49   41.49   41.49   41.49   41.49
   41.49   41.48   41.48   41.48   41.48   41.47   41.47   41.47   41.47   41.46
   41.46   41.46   41.46   41.46   41.46   41.46   41.47   41.47    41.7    41.7
   41.86   41.88   41.88   41.88   41.84    41.8    41.8    41.8    41.8   41.83
   41.76
   41.63    41.5   41.47    40.8   40.79   41.08    41.1   41.23   41.24   40.53
   40.49   40.03   40.36   41.27   40.69    40.6   40.51   39.59   39.59   39.59
   39.59   39.58   39.58   39.58   39.58   39.57   39.57   39.57   39.57   39.56
   39.57   39.59   41.14   41.21   41.22   41.23   41.25   41.29   41.26   41.26
   39.17   40.99   41.21   41.21   41.53   41.62   41.62   41.67   41.75   41.75
   41.76
  4597.9  4758.3  4802.8  4819.6  4819.8  4851.8  4853.8  4888.2  4890.9  4939.1
  4941.2  4966.2  4973.2  4983.9 4984.51  4984.6  4984.7 4985.79  4985.9 4986.01
  4986.8  4990.6  4991.4  4995.7  4995.9  5002.6  5003.6  5004.3  5015.5  5019.6
 5019.69  5019.8  5026.7 5027.99  5028.1 5028.21  5028.6  5028.7  5044.4  5044.7
  5089.5  5095.2  5095.3  5095.4  5119.4  5144.2  5144.6  5162.5  5190.1  5190.4
  5192.6
   41.72   41.59   41.56   41.94   41.94   41.83   41.83   41.81    41.8   41.59
   41.58   41.53   41.52   41.49   41.49   41.49   41.49   41.49   41.49   41.49
   41.49   41.48   41.48   41.48   41.48   41.47   41.47   41.47   41.47   41.46
   41.46   41.46   41.46   41.46   41.46   41.46   41.47   41.47    41.7    41.7
   41.86   41.88   41.88   41.88   41.84    41.8    41.8    41.8   41.84   41.84
   41.85
   41.72   41.59   41.56   40.89   40.88   41.17   41.19   41.32   41.33   40.62
   40.58   40.12   40.45   41.36   40.78   40.69    40.6   39.68   39.68   39.68
   39.68   39.67   39.67   39.67   39.67   39.66   39.66   39.66   39.66   39.65
   39.66   39.68   41.23    41.3   41.31   41.32   41.34   41.38   41.35   41.35
   39.26   41.08    41.3    41.3   41.62   41.71   41.71   41.76   41.84   41.84
   41.85
Pier Skew, UpSta & Num, DnSta & Num=,4996.6, 2 ,4996.6, 2 , 0 , 0 , 0 ,,
       1       1
   28.99   40.58
       1       1
   29.08   40.67
Pier Skew, UpSta & Num, DnSta & Num=,5010.4, 2 ,5010.4, 2 , 0 , 0 , 0 ,,
       1       1
   35.15   40.57
       1       1
   35.24   40.66
BR Coef= 1 , 1 , 0 ,1.25, 0 ,,,0.8,0,2,0,
Wspro=,,,, 1 ,,,, 0 ,,,, 0 ,,,,-1 ,-1 ,-1 , 0 , 0 , 0 , 0 , 0
BC Design=,, 0 ,, 0 ,,,,,,
BR U #Sta/Elev= 51
  4597.9   41.63  4758.3    41.5  4802.8   41.47  4819.6    40.8  4819.8   40.79
  4851.8   41.08  4853.8    41.1  4888.2   41.23  4890.9   41.24  4939.1   40.53
  4941.2   40.49  4966.2   40.03  4973.2   40.36  4983.9   41.27 4984.51   40.69
  4984.6    40.6  4984.7   40.51 4985.79   39.46  4985.9   39.36 4986.01   39.25
  4986.8    38.5  4990.6   36.37  4991.4   35.92  4995.7   33.74  4995.9   29.99
  5002.6   30.01  5003.6   29.91  5004.3   33.68  5015.5   38.63  5019.6   39.55
 5019.69   39.57  5019.8   39.59  5026.7   41.14 5027.99   41.21  5028.1   41.22
 5028.21   41.23  5028.6   41.25  5028.7   41.29  5044.4   41.26  5044.7   41.26
  5089.5   39.17  5095.2   40.99  5095.3   41.21  5095.4   41.21  5119.4   41.53
  5144.2   41.62  5144.6   41.62  5162.5   41.67  5190.1   41.75  5190.4   41.75
  5192.6   41.76
BR U #Mann= 5
 4597.90     0.2  4758.3     0.1  4986.8    0.02  5015.5     0.1  5162.5     0.2
BR U Banks=4986.80,5015.50
BR D #Sta/Elev= 51
  4597.9   41.72  4758.3   41.59  4802.8   41.56  4819.6   40.89  4819.8   40.88
  4851.8   41.17  4853.8   41.19  4888.2   41.32  4890.9   41.33  4939.1   40.62
  4941.2   40.58  4966.2   40.12  4973.2   40.45  4983.9   41.36 4984.51   40.78
  4984.6   40.69  4984.7    40.6 4985.79   39.55  4985.9   39.45 4986.01   39.34
  4986.8   38.59  4990.6   36.46  4991.4   36.01  4995.7   33.83  4995.9   30.08
  5002.6    30.1  5003.6      30  5004.3   33.77  5015.5   38.72  5019.6   39.64
 5019.69   39.66  5019.8   39.68  5026.7   41.23 5027.99    41.3  5028.1   41.31
 5028.21   41.32  5028.6   41.34  5028.7   41.38  5044.4   41.35  5044.7   41.35
  5089.5   39.26  5095.2   41.08  5095.3    41.3  5095.4    41.3  5119.4   41.62
  5144.2   41.71  5144.6   41.71  5162.5   41.76  5190.1   41.84  5190.4   41.84
  5192.6   41.85
BR D #Mann= 5
 4597.90     0.2  4758.3     0.1  4986.8    0.02  5015.5     0.1  5162.5     0.2
BR D Banks=4986.80,5015.50

Type RM Length L Ch R = 1 ,411.7,4.9,4.9,4.9
XS GIS Cut Line= 4
      3137038.61     13859515.84      3137204.25     13859599.11
      3137547.32     13859613.31      3137613.08     13859608.41
BEGIN DESCRIPTION:
Downstream Section of Bridge/Culvert/Weir
END DESCRIPTION:
#Sta/Elev= 27
  4597.9   41.53  4758.3    41.4  4802.8   41.37  4819.8   40.69  4853.8      41
  4890.9   41.14  4939.1   40.43  4966.2   39.93  4973.2   40.26  4983.9   41.17
  4986.8    38.4  4991.4   35.82  4995.7   33.64  4995.9   29.89  5002.6   29.91
  5003.6   29.81  5004.3   33.58  5015.5   38.53  5026.7   41.04  5028.7   41.19
  5044.7   41.16  5089.5   39.07  5095.2   40.89  5095.3   41.11  5119.4   41.43
  5162.5   41.57  5192.6   41.66
#Mann= 5 , 1 , 0
 4597.90     0.2       0  4758.3     0.1       0  4986.8    0.02       0
  5015.5     0.1       0  5162.5     0.2       0
#XS Ineff= 2 , 0
       0    4975    41.3    5030       0    41.3
Bank Sta=4986.80,5015.50
Exp/Cntr=0.5,0.3

Type RM Length L Ch R = 1 ,406.8,0,0,0
XS GIS Cut Line= 4
      3137037.11     13859618.87      3137368.85     13859613.53
      3137442.66     13859614.93      3137572.49     13859621.45
BEGIN DESCRIPTION:
Cross Section 406.8
END DESCRIPTION:
#Sta/Elev= 29
  4614.1   47.13  4629.1   46.94  4644.1   44.64  4659.1   41.71  4674.1   41.06
  4689.1   41.07  4734.1   42.94  4764.1   42.66  4804.1   40.86  4824.1   40.95
  4854.1   40.41  4914.1   40.79 4921.43   40.62 4947.43   41.07 4980.83   38.81
 4982.23   38.82 4987.73   36.23 4992.93    33.8 4993.43   30.06 5004.63   29.73
 5005.73   29.76 5007.03   33.75 5012.03   35.75 5018.83   38.55 5021.83   39.14
 5027.53   37.46 5063.73    41.3  5134.7   40.96  5149.7   41.49
#Mann= 3 , 1 , 0
 4614.10     0.1       0 4982.23    0.02       0 5018.83     0.1       0
Bank Sta=4982.23,5018.83
Exp/Cntr=0.3,0.1

Chan Stop Cuts=-1
